--- LFFILESCK.prj (project) ---

Proj Title=LFFILESCK
Current Plan=p01
Default Exp/Contr=0,0
English Units
Geom File=g01
Flow File=f01
Plan File=p01
BEGIN DESCRIPTION:
----------MODEL BY WOOD PLC 2022----------
AFH study
Randolph County, WV
HEC-RAS Version: RAS 6.2
Vertical Datum: NAVD88
Projection: NAD 1983 StatePlane West Virginia S FIPS 4702 (US Feet)
Terrain: 1-meter LIDAR (FEMA Region III 3DEP collected 2016-2018)
Land Use: 2019 NLCD
Hydrologic Method:
WV SIR2010-5033 regression equations
Additional Model Notes:
Main stem is FILESCK/RFFILESCK
END DESCRIPTION:
DSS Export Rating Curves= 0
DSS Export Rating Curve Sorted= 0
DSS Export Volume Flow Curves= 0
DXF OffsetX= 0
DXF OffsetY= 0
DXF ScaleX= 0
DXF ScaleY= 0

--- LFFILESCK.p01 (plan) ---

Plan Title=Floodplain
Program Version=6.20
Short Identifier=Floodplain
Geom File=g01
Flow File=f01
Subcritical Flow
K Sum by GR= 0
Std Step Tol= 0.01
Critical Tol= 0.01
Num of Std Step Trials= 20
Max Error Tol= 0.3
Flow Tol Ratio= 0.001
Split Flow NTrial= 30
Split Flow Tol= 0.02
Split Flow Ratio= 0.02
Log Output Level= 0
Friction Slope Method= 1
Unsteady Friction Slope Method= 2
Unsteady Bridges Friction Slope Method= 1
Parabolic Critical Depth
Global Vel Dist= 0 , 0 , 0
Global Log Level= 0
CheckData=True
Encroach Param=-1 ,0,0, 0
Mapping Interval=1HOUR
Computation Time Step Use Courant=        0
Computation Time Step Use Time Series=    0
Computation Time Step Count To Double=0
Computation Time Step Max Doubling=0
Computation Time Step Max Halving=0
Computation Time Step Residence Courant=0
Run HTab= 0
Run UNet= 0
Run Sediment= 0
Run PostProcess= 0
Run WQNet= 0
Run RASMapper=-1
UNET Theta= 0
UNET Theta Warmup= 0
UNET ZTol= 0
UNET ZSATol= 0
UNET MxIter= 0
UNET Max Iter WO Improvement= 0
UNET MaxInSteps= 0
UNET DtIC= 0
UNET DtMin= 0
UNET MaxCRTS= 0
UNET WFStab= 0
UNET SFStab= 0
UNET WFX= 1
UNET SFX= 1
UNET Gravity=32.174
UNET 1D Methodology=Finite Difference
UNET DSS MLevel= 1
UNET Pardiso=0
UNET DZMax Abort= 0
UNET Use Existing IB Tables= 0
UNET Froude Reduction=False
UNET Froude Limit= 0
UNET Froude Power= 0
UNET D1 Cores= 0
UNET WindReference=Eulerian
UNET WindDragFormulation=Hsu (1988)
UNET D2 Coriolis=0
UNET D2 Cores= 0
UNET D2 Theta= 1
UNET D2 Theta Warmup= 1
UNET D2 Z Tol= 0.01
UNET D2 Volume Tol= 0.01
UNET D2 Max Iterations= 20
UNET D2 Equation= 0
UNET D2 RampUpFraction=0.1
UNET D2 TimeSlices= 1
UNET D2 Turbulence Formulation=Non-Conservative (original)
UNET D2 Eddy Viscosity=0.3
UNET D2 Transverse Eddy Viscosity=0.1
UNET D2 Smagorinsky Mixing=0
UNET D2 BCVolumeCheck=0
UNET D2 Cores=0
UNET D2 SolverType=PARDISO (Direct)
UNET D2 Minimum Iterations= 2147483647
UNET D2 Maximum Iterations= 2147483647
UNET D2 Restart Number= 10
UNET D2 Relaxation Coeff=1.3
UNET D2 SOR Precondition Iterations= 10
UNET D2 ILUT Maximum Fill= 8
UNET D2 ILUT Tolerance=1E-08
UNET D1D2 MaxIter= 0
UNET D1D2 ZTol=0.01
UNET D1D2 QTol=0.1
UNET D1D2 MinQTol=1
Write IC File= 0
Write IC File at Fixed DateTime=0
Write IC File at Sim End=0
Echo Input=False
Echo Parameters=False
Echo Output=False
Write Detailed= 0
HDF Write Warmup=0
HDF Write Time Slices=0
HDF Flush=0
HDF Compression= 1
HDF Chunk Size= 1
HDF Spatial Parts= 1
HDF Use Max Rows=0
HDF Fixed Rows= 1
Calibration Method= 0
Calibration Iterations= 20
Calibration Max Change=0.05
Calibration Tolerance=0.2
Calibration Maximum=1.5
Calibration Minimum=0.5
Calibration Optimization Method= 1
WQ AD Non Conservative
WQ ULTIMATE=-1
WQ Max Comp Step=1HOUR
WQ Output Interval=15MIN
WQ Output Selected Increments= 0
WQ Output face flow=0
WQ Output face velocity=0
WQ Output face area=0
WQ Output face dispersion=0
WQ Output cell volume=0
WQ Output cell surface area=0
WQ Output cell continuity=0
WQ Output cumulative cell continuity=0
WQ Output face conc=0
WQ Output face dconc_dx=0
WQ Output face courant=0
WQ Output face peclet=0
WQ Output face adv mass=0
WQ Output face disp mass=0
WQ Output cell mass=0
WQ Output cell source sink temp=0
WQ Output nsm pathways=0
WQ Output nsm derived pathways=0
WQ Create Restart=0
WQ Fixed Restart=0
WQ System Summary=0
WQ Write To DSS=0
Sorting and Armoring Iterations= 10
XS Update Threshold= 0.02
Bed Roughness Predictor= 0
Hydraulics Update Threshold= 0.02
Energy Slope Method= 1
Volume Change Method= 1
Sediment Retention Method= 0
Sediment TS Multiplier= 1
Warm Up Method= 0
XS Weighting Method= 0
Number of US Weighted Cross Sections= 1
Number of DS Weighted Cross Sections= 1
Upstream XS Weight=0
Main XS Weight=1
Downstream XS Weight=0
Number of DS XS's Weighted with US Boundary= 1
Upstream Boundary Weight= 1
Weight of XSs Associated with US Boundary= 0
Number of US XS's Weighted with DS Boundary= 1
Downstream Boundary Weight= 0.5
Weight of XSs Associated with DS Boundary= 0.5
Percentile Method= 0
Sediment Output Level= 3
Mass or Volume Output= 0
Output Increment Type= 1
Profile and TS Output Increment= 1
Transport Output Increment 1
XS Output Flag= 0
XS Output Increment= 10
Read HDF5 Sediment Hotstart= 0
Sediment Hotstart Type= 0
Write Gradation File= 0
Read Gradation Hotstart= 0
Write HDF5 File= 1
Write Binary Output= 1
Write DSS Sediment File= 0
DSS Sediment Output Type= 1
SV Curve= 0
Specific Gage Flag= 0
Subcell Erosion Methods= 0
Subcell Deposition Methods= 0
Advection Scheme= 1
Matrix Solver= 0
Implicit Weighting Factor= 1
Maximum Outer Loop Convergence Iterations= 5
Convergence Maximum Absolute= 0.001
Convergence RMSE= 0.0001
Grain Fractions Max Abs Error= 0.001
Max Subgrid Regions= 1
Max Subgrid Length Scale= 3.402823E+38
Initial Layer Thickness= 3.402823E+38
Min Layer Thickness= 3.402823E+38
Max Layer Thickness= 3.402823E+38
Number of Layers= 5

--- LFFILESCK.f01 (steady flow) ---

Flow Title=Flow
Program Version=6.20
Number of Profiles= 1
Profile Names=P100yr
River Rch & RM=LFFILESCK,Main,16036
     857
River Rch & RM=LFFILESCK,Main,11876
    1030
River Rch & RM=LFFILESCK,Main,10757
    1210
River Rch & RM=LFFILESCK,Main,5047
    1360
Boundary for River Rch & Prof#=LFFILESCK,Main            , 1
Up Type= 0
Dn Type= 3
Dn Slope=0.01497
DSS Import GetInterval= 0
DSS Import GetPeak= 0
DSS Import FillOption= 0

--- LFFILESCK.g01 (geometry) ---

Geom Title=Geometry
Program Version=6.20

River Reach=LFFILESCK       ,Main
Reach XY= 30
2311737.00972155670318.6368971772311957.76500002670120.881000012
2311917.07400002669645.2820000052311278.48700002669131.428000003
2311086.95500003668017.0970000182310457.74400003667731.288000017
2310094.57800002667414.0509999992309847.24400002667504.371000022
2309504.45100002667409.863000005      2309148.22667452.983999997
2308965.90300001667622.9960000072308169.34200002667638.472000018
2307281.99900001666936.5120000092306481.67299999666578.381999999
2306310.88200001666284.0390000052305777.38899998666276.695999995
2305627.94600002666373.324000016     2304705.839666058.334000021
2304353.31000005665773.2410000262303613.32700005665867.831000015
2303192.20899999 665643.23800002     2302657.149665502.250000015
2302410.65000001665575.5080000012302217.91400003665762.510000005
2301597.15185347665593.0757327042301344.50699998665655.881000012
2301091.17700005665564.1660000092300386.34608085665558.558434159
2299808.88200001665342.8320000022299452.53093168665072.852208212

Type RM Length L Ch R = 1 ,16036   ,31.9,35.3,38.6
XS GIS Cut Line= 5
 2311926.4929505670456.701425856 2311791.5228368670371.698584684
 2311741.3543004670336.2759348182311732.27389828670299.409402902
2311627.36462561670211.749385274
#Sta/Elev= 30
       0 2475.12    12.2 2468.04    31.1 2458.06    59.5 2443.93   111.6 2415.04
   131.9 2400.64   140.6 2393.66   144.6 2390.16   149.2 2384.83     154 2380.42
   158.7 2376.92   163.6 2375.74   183.2 2375.34     193 2373.41   209.6 2374.68
   224.1 2373.47  227.352372.684   236.5 2371.59   244.7 2371.61  249.742372.685
   252.9 2374.15   260.5 2375.83   263.4 2376.98   269.1 2380.02   287.3 2391.77
   293.6 2393.98   316.4 2396.59   331.5  2399.3   349.7 2399.64   395.6 2402.36
#Mann= 5, -1 ,  0
       0     0.1       0      80    0.06       0  199.51     0.1       0
  227.35   0.045       0  249.74     0.1       0
Bank Sta=227.35,249.74
XS Rating Curve= 0 ,0
Exp/Cntr=0.3,0.1

Type RM Length L Ch R = 1 ,16000   ,40.5,38.8,48.4
XS GIS Cut Line= 6
2311976.87859864670433.483880595 2311765.8171805670339.327601147
2311774.15076119670289.0572918362311785.72302802670252.565364664
 2311803.9277785670224.6772362572311572.17756772670120.070724811
#Sta/Elev= 30
       0 2500.63    13.9 2489.72    40.1 2471.74    55.2 2462.46    80.2 2449.05
   119.1 2429.58     141 2416.43     163 2401.08   182.4 2385.92   197.5 2375.23
   237.3 2374.38  253.27  2371.2   265.6 2369.82   269.7 2370.28  271.48  2371.2
   277.9 2374.29   298.7 2373.38   321.7 2373.76   353.7 2373.05   362.2 2377.81
   365.2 2378.41     371  2377.5   380.3 2379.87   388.5 2383.76   397.3 2389.85
   407.5 2392.22   524.6 2399.67   550.9 2402.08   581.6 2403.88   607.9  2406.6
#Mann= 7, -1 ,  0
       0     0.1       0     120    0.06       0  253.27   0.045       0
  271.48    0.06       0  403.67     0.1       0  443.67    0.06       0
  513.67    0.07       0
Bank Sta=253.27,271.48
XS Rating Curve= 0 ,0
Exp/Cntr(USF)=0,0
Exp/Cntr=0.3,0.1

Type RM Length L Ch R = 1 ,15962   ,130.1,122.6,100.7
XS GIS Cut Line= 6
2312011.30191003670424.9377105682311800.24049189 670330.78143112
2311805.61699556670294.758856533 2311814.7570518670259.273932314
2311834.98466158670225.1056000192311584.53986044670105.319893282
#Sta/Elev= 30
       0 2520.16    29.4 2496.59    69.2 2468.33    95.5 2452.85   135.4  2433.4
   161.2 2419.64   200.6 2389.62   218.1 2377.88   226.8 2374.17   253.6 2372.41
  263.462369.893   269.1 2368.91   285.6 2368.88  291.682369.892   306.5 2372.44
   315.8 2371.63   325.3  2372.5   351.6 2371.85   369.3  2372.6   373.8 2373.91
   382.1 2377.97   387.1 2377.67   395.9  2378.8   415.1 2387.96   430.1 2391.34
   484.6 2396.03   506.8 2396.62   550.1 2399.71   584.9 2402.72   621.7 2407.16
#Mann= 5, -1 ,  0
       0     0.1       0     100    0.06       0  263.46   0.045       0
  291.68    0.06       0  544.05    0.07       0
#XS Ineff= 2 , 0
                          338.42          2378.7
Permanent Ineff=
       F       F
Bank Sta=263.46,291.68
XS Rating Curve= 0 ,0
Exp/Cntr(USF)=0,0
Exp/Cntr=0.3,0.1

Type RM Length L Ch R = 1 ,15839   ,313,308.5,300.5
XS GIS Cut Line= 3
2312082.63298125670336.0407013222311852.36401744670182.979566558
2311589.58649404670086.808411087
#Sta/Elev= 30
       0 2516.27    79.8 2462.01   145.2 2421.75     177 2398.38   197.1 2380.53
   207.5 2369.09  211.63 2366.31   214.7  2365.3   228.7 2364.96   233.5 2366.32
   237.5 2368.57   240.4 2369.17   247.9 2369.56   257.7 2368.66   266.4 2370.53
   285.2 2370.83   302.3 2373.01     315 2373.45   323.6 2375.95   336.3 2382.02
   343.5 2384.49   377.8 2393.08   394.7 2396.13   421.5 2398.35   440.2 2398.57
   506.7 2405.46   515.2 2405.69   536.5 2408.56   546.2  2410.7   556.3  2411.6
#Mann= 6, -1 ,  0
       0     0.1       0  211.63   0.045       0   233.5     0.1       0
     270    0.06       0   486.5    0.07       0   546.5    0.06       0
#XS Ineff= 2 , 0
                          247.72         2373.01
Permanent Ineff=
       F       F
Bank Sta=211.63,233.5
XS Rating Curve= 0 ,0
Exp/Cntr(USF)=0,0
Exp/Cntr=0.3,0.1

Type RM Length L Ch R = 1 ,15531   ,503.1,492.3,480.7
XS GIS Cut Line= 4
2312209.71766943670130.2169964722312003.70138522669933.865544149
2311879.77710183669933.3255391482311561.39970019669968.445927891
#Sta/Elev= 30
       0 2500.88    18.8 2496.82    30.1 2492.62   111.7  2448.5   140.7 2430.85
   167.9 2417.54   206.6 2402.12   234.2 2382.38   262.1 2365.95   272.9 2364.51
   284.6 2366.25   320.7 2363.55  342.712359.822   352.1 2358.75  362.562359.823
   372.1 2363.55   392.1 2365.18   412.1 2368.67   444.3 2368.63   452.4 2371.08
   472.5 2373.75   488.6 2378.44   512.8 2377.94     524 2385.42   532.9 2388.91
   571.1 2398.71   603.8 2405.09   673.7 2410.81   705.9 2422.19   728.8  2427.9
#Mann= 7, -1 ,  0
       0     0.1       0   334.6    0.06       0  342.71   0.045       0
  362.56    0.06       0  528.52     0.1       0  628.52    0.07       0
  728.52     0.1       0
Bank Sta=342.71,362.56
XS Rating Curve= 0 ,0
Exp/Cntr=0.3,0.1

Type RM Length L Ch R = 1 ,15038   ,405.1,398.8,394.7
XS GIS Cut Line= 4
2312024.79833403669420.4043290142311776.54841554669500.106216838
2311699.23891093 669632.115128042311503.91779205669818.176980293
#Sta/Elev= 30
       0 2476.96    10.7 2472.67    71.1 2441.35    80.5 2438.92    93.3 2430.61
   118.3 2418.65   151.9 2404.72   172.9 2398.49   185.6 2393.49   202.3 2384.51
   210.7 2381.72   223.7 2372.41   248.5 2358.62   260.7  2352.8   270.6 2349.49
  279.392347.775   289.8 2346.56  302.022347.776   320.3 2353.03   343.6 2352.33
   396.3 2356.68   455.8 2356.12   484.8 2361.92     508 2361.77   517.4 2363.76
   532.6 2364.22   560.2 2375.05   600.2 2389.02   648.6 2408.78   683.5  2420.9
#Mann= 5, -1 ,  0
       0     0.1       0  279.39   0.045       0  302.02    0.05       0
  473.71    0.06       0  513.71     0.1       0
Bank Sta=279.39,302.02
XS Rating Curve= 0 ,0
Exp/Cntr=0.3,0.1

Type RM Length L Ch R = 1 ,14639   ,59.4,59.6,59.2
XS GIS Cut Line= 6
2311797.98712902668969.8837489342311462.73110483669141.213325967
2311485.99808443669197.2655949962311477.53736458669297.736643256
2311551.56866329669377.0558918822311321.01404729669739.809255598
#Sta/Elev= 30
       0 2456.67    87.4 2446.64   104.9 2443.22   119.7 2436.57   131.6 2435.07
   150.3 2429.06   182.2 2415.31   226.3 2389.48   265.4 2362.89   289.5  2348.6
     310 2345.74   361.4 2338.59   462.7 2340.45  475.712338.521   483.9 2337.47
   502.22338.527   512.4 2341.24   571.2 2341.78   624.1 2344.69   688.2 2345.17
   740.3  2347.5   771.5 2350.19   797.5 2355.76   835.4    2358   847.5 2364.99
   877.7 2375.92   915.7 2386.95   939.4 2392.17     982 2406.91  1079.9 2445.16
#Mann= 8, -1 ,  0
       0     0.1       0     310    0.05       0   376.5    0.06       0
   386.5    0.05       0  475.71   0.045       0   502.2    0.05       0
   800.1    0.06       0   920.1     0.1       0
#XS Ineff= 2 , 0
          465.33  2346.1
Permanent Ineff=
       F       F
Bank Sta=475.71,502.2
XS Rating Curve= 0 ,0
Exp/Cntr(USF)=0,0
Exp/Cntr=0.3,0.1

Type RM Length L Ch R = 1 ,14580   ,290.7,306.3,319.1
XS GIS Cut Line= 6
2311748.02742436668968.6347563182311412.77140017 669139.96433335
2311436.03837977669196.0166023792311427.57765991669296.487650639
2311501.60895863669375.8068992652311271.05434262669738.560262982
#Sta/Elev= 30
       0 2441.31    50.8 2436.55    68.7  2432.1    80.7 2426.68    94.2 2425.69
   101.4 2423.51   178.7 2384.77   242.4  2347.1   279.7 2343.87   324.3 2337.53
   427.7 2338.91   439.8 2337.45   447.8 2336.16  465.332337.434     480 2341.67
   549.8  2342.1   561.5 2343.51   568.1 2342.34   624.6 2342.71   727.6  2346.7
   776.7 2357.43   808.1 2358.91   831.7 2371.28   860.3 2380.56   881.1 2385.54
   901.3 2387.87   912.9 2392.67   955.1  2403.7  1002.4 2423.62  1079.9 2451.65
#Mann= 9, -1 ,  0
       0     0.1       0     310    0.05       0     320    0.06       0
   439.8   0.045       0  465.33    0.05       0  549.71    0.06       0
  604.55    0.05       0   720.1    0.06       0   920.1     0.1       0
Bank Sta=439.8,465.33
XS Rating Curve= 0 ,0
Exp/Cntr(USF)=0,0
Exp/Cntr=0.3,0.1

Type RM Length L Ch R = 1 ,14274   ,295.5,295.6,296.5
XS GIS Cut Line= 4
2311725.24415369668932.5133511162311403.92418964668959.568235488
2311231.25707863669011.9900364532310943.26318354669193.832448139
#Sta/Elev= 30
       0 2425.27     9.1 2423.91    17.1  2420.9    53.3 2411.89    61.8 2407.56
    77.3 2404.92   153.6 2368.02   189.7 2353.93   217.8 2344.59     274 2340.53
   294.1 2337.25   347.3 2337.69     364  2332.2   429.4  2333.4  466.332330.357
   480.7 2329.39  490.362330.358   511.8 2343.68   520.7 2347.85   572.7 2362.96
   581.4 2364.33   590.1 2368.37   607.5 2369.04   619.1 2374.13   643.7 2375.55
   648.5 2378.08   692.4 2389.99   722.4 2400.67     796 2421.29   843.5 2438.44
#Mann= 8, -1 ,  0
       0     0.1       0     270    0.05       0  362.46     0.1       0
  466.33   0.045       0  490.36    0.05       0  492.46     0.1       0
  582.91    0.06       0  682.91     0.1       0
Bank Sta=466.33,490.36
XS Rating Curve= 0 ,0
Exp/Cntr=0.3,0.1

Type RM Length L Ch R = 1 ,13978   ,432.5,438.3,441.9
XS GIS Cut Line= 4
2311626.96644917668589.6308023852311278.09022283668707.923723775
2311158.93562293668743.7929222022310800.69873651668853.903053945
#Sta/Elev= 30
       0 2449.76      41  2430.2    70.5 2413.14      79 2406.22    87.4 2403.86
   142.3 2368.07   150.8 2360.25   163.4 2357.92   184.8 2345.55   206.9 2340.34
   239.5 2337.19   391.3 2330.07  410.132323.934   416.3 2322.33   430.72323.936
     471 2326.14   491.5 2330.02   512.4 2340.43   545.9 2362.23   579.4 2373.15
   601.8 2373.62   617.1 2382.12     638 2383.57   675.7 2393.95   688.2 2401.07
   734.2 2413.02   759.3 2421.74   780.3 2423.52   809.6 2433.45   867.6  2448.5
#Mann= 8, -1 ,  0
       0     0.1       0     180    0.07       0     280    0.06       0
  378.39     0.1       0  410.13   0.045       0   430.7     0.1       0
  488.39    0.06       0  592.82     0.1       0
Bank Sta=410.13,430.7
XS Rating Curve= 0 ,0
Exp/Cntr=0.3,0.1

Type RM Length L Ch R = 1 ,13540   ,553.2,538.8,520.6
XS GIS Cut Line= 4
2311600.94257866668264.7001567172311270.76576319668323.505314164
 2311102.8996013668311.1326998572310745.43189572668449.294000605
#Sta/Elev= 30
       0 2534.62      17 2525.13    37.3 2511.32    45.5 2509.61    65.8 2496.66
    90.2 2484.12   151.1 2441.75   183.3 2422.31   191.7 2415.56     208 2409.13
   216.1 2401.39   228.3 2392.74   305.5 2345.65   317.7 2332.96   325.8 2326.77
     346    2323   390.1 2321.88  415.622314.675   422.1 2313.75  443.942314.674
   466.3 2317.77   522.8 2317.56   536.6 2330.42   549.5 2337.55   588.1 2351.22
   605.2 2353.63   622.4 2353.22   635.3 2358.82   682.4 2371.49   886.9  2418.9
#Mann= 5, -1 ,  0
       0     0.1       0  415.62   0.045       0  443.94     0.1       0
  445.37    0.06       0  643.69     0.1       0
#XS Ineff= 2 , 0
                          467.92         2331.98
Permanent Ineff=
       F       F
Bank Sta=415.62,443.94
XS Rating Curve= 0 ,0
Exp/Cntr=0.3,0.1

Type RM Length L Ch R = 1 ,13001   ,481.7,483.5,485.4
XS GIS Cut Line= 4
     2311089.984      667514.0292310933.24337354 667821.13632499
2310851.46400109668011.0299985752310661.14636923668306.273368562
#Sta/Elev= 30
       0 2538.64    21.5 2534.44    72.1 2506.84    97.8 2489.96   111.3 2477.35
   124.8 2472.98   143.4 2457.28   192.2 2424.97   208.8 2411.49     304 2349.63
   312.9 2341.14   322.4 2326.97   348.7 2310.26   366.9 2305.01   418.9 2306.67
   442.52300.875   455.2 2299.59     4662300.873   488.6 2309.03   514.7 2308.13
   529.5 2303.91   545.2 2305.03   587.1 2322.28   616.3 2322.72   625.5 2328.98
   673.1 2340.82   739.7 2370.43   807.2 2389.47   847.7 2405.83   902.8 2420.28
#Mann= 5, -1 ,  0
       0     0.1       0   442.5   0.045       0     466     0.1       0
  494.79    0.06       0  691.55     0.1       0
Bank Sta=442.5,466
XS Rating Curve= 0 ,0
Exp/Cntr=0.3,0.1

Type RM Length L Ch R = 1 ,12517   ,340.7,343.5,345.7
XS GIS Cut Line= 4
2310661.43067278667444.3469718672310480.49603543667669.277988233
2310402.05359352667806.7352579282310270.06740648      668114.738
#Sta/Elev= 30
       0 2489.16    15.7  2474.8    26.7 2471.08    31.9 2467.69    42.1 2458.29
    52.7 2450.26   135.2 2396.42   170.5 2369.45   229.1 2330.73   238.1 2323.66
   242.3 2321.53   254.7 2319.47   274.6 2304.56   293.2 2292.26   325.4 2293.05
  336.852292.162   357.6 2291.05     370 2292.17   376.8  2293.7   389.9  2291.6
   403.7 2293.77   438.4 2294.04   453.9 2296.01   459.4  2298.4   492.3 2320.31
   508.1 2328.87   558.4 2349.66   641.1 2379.64     702 2405.79     782 2444.07
#Mann= 4, -1 ,  0
       0     0.1       0  336.85   0.045       0     370    0.06       0
  476.94     0.1       0
Bank Sta=336.85,370
XS Rating Curve= 0 ,0
Exp/Cntr=0.3,0.1

Type RM Length L Ch R = 1 ,12174   ,320.2,297.9,282.3
XS GIS Cut Line= 4
2310468.64557289667357.2790475752310213.63839356667479.447480302
2310102.98941713667618.264398779     2309980.496      667941.622
#Sta/Elev= 30
       0 2444.49    71.5 2405.64    92.3 2390.89   168.2 2344.72   200.1 2322.76
   235.6 2302.34   266.6 2288.23     285    2288  315.632283.506  335.412283.502
   344.8 2286.14   364.7 2286.32   371.9 2285.36   382.2 2281.55   394.2 2283.78
   428.2 2282.98   458.7 2286.29   467.7 2292.19   484.8 2307.77   502.1 2318.27
   548.5 2338.62   581.1 2354.49   621.7 2367.13   647.8 2379.65   694.3 2407.13
   719.1 2416.92   724.3 2420.23   732.9 2420.79   784.2  2441.7   806.1  2447.3
#Mann= 4, -1 ,  0
       0     0.1       0  315.63   0.045       0  335.41    0.06       0
  480.28     0.1       0
#XS Ineff= 2 , 0
                          354.23         2292.93
Permanent Ineff=
       F       F
Bank Sta=315.63,335.41
XS Rating Curve= 0 ,0
Exp/Cntr=0.3,0.1

Type RM Length L Ch R = 1 ,11876   ,40.3,42.9,42.7
XS GIS Cut Line= 6
2310059.90033273666952.0483212452309793.08624308667323.841354009
2309921.06943712667418.6722748972309975.03825389667462.618311406
2310096.08260006 667535.090722492309926.66079204667897.625762786
#Sta/Elev= 30
       0 2390.81    52.2 2366.79   119.8 2340.66   144.4  2337.6   166.8 2328.52
   188.8 2324.38   208.5 2315.54   238.1 2309.06   310.1 2302.24   341.7 2288.72
   376.2 2282.83   416.1 2282.39   453.5 2277.76   606.7 2279.17  616.962275.827
     621 2274.44  646.792275.825   652.6 2279.49     659 2279.86     837 2282.82
   891.9 2280.61   904.5 2287.21   928.5 2307.94   944.8 2318.91   993.4 2339.91
  1003.8  2348.5  1024.3 2356.04  1092.1 2386.91  1163.2 2423.46  1227.9 2449.78
#Mann= 5, -1 ,  0
       0     0.1       0  616.96   0.045       0  646.79     0.1       0
  647.01    0.06       0  937.74     0.1       0
#XS Ineff= 2 , 0
          602.64 2289.32
Permanent Ineff=
       F       F
Bank Sta=616.96,646.79
XS Rating Curve= 0 ,0
Exp/Cntr(USF)=0,0
Exp/Cntr=0.3,0.1

Type RM Length L Ch R = 1 ,11833   ,307,317.3,326
XS GIS Cut Line= 6
2310031.06733818 666979.363789772309764.25324852667351.156822534
2309892.23644257667445.9877434212309946.20525933 667489.93377993
2310067.24960551667562.4061910152309897.82779749667924.941231311
#Sta/Elev= 30
       0 2373.34    76.2 2344.95    86.1  2339.7   103.7 2336.84     128 2328.93
   140.9 2327.72   174.9 2314.47   203.9 2308.57   268.6 2302.46   293.2 2290.22
   326.3 2284.13   450.9 2277.01   464.8 2274.53     612  2277.7  620.532274.682
   630.6 2273.28  640.942274.654     659 2279.58   685.4  2276.6   703.2 2279.05
     810 2283.16   835.2 2281.12   861.7  2281.9   901.3 2312.99   919.1 2324.33
   980.9 2351.07   994.6 2361.88  1061.8 2391.95    1124 2423.12  1227.9 2468.58
#Mann= 7, -1 ,  0
       0     0.1       0     440    0.06       0  495.93     0.1       0
  604.09    0.06       0  620.53   0.045       0  640.94    0.06       0
  907.74     0.1       0
#XS Ineff= 2 , 0
          605.01 2289.57  656.92         2289.39
Permanent Ineff=
       F       F
Bank Sta=620.53,640.94
XS Rating Curve= 0 ,0
Exp/Cntr(USF)=0,0
Exp/Cntr=0.3,0.1

Type RM Length L Ch R = 1 ,11516   ,411.2,405.8,400.4
XS GIS Cut Line= 4
2309536.42203941667054.4622218832309630.93987075 667419.06291578
2309610.88079035667516.1685788642309645.42478084667866.858494393
#Sta/Elev= 30
       0 2327.15    56.5 2308.17    97.8 2301.23   142.5 2299.02   156.3  2296.8
   188.8 2296.94   217.7  2295.3   263.1 2285.41   267.3 2283.66   284.2 2273.07
     381 2271.01     387 2269.96  393.282266.769   397.7 2265.75   407.9 2265.61
   419.7 2265.75  424.712266.771   431.6 2269.73   434.9 2270.14   444.2 2268.89
   476.8 2270.58   488.9 2274.06   496.9 2275.09     505 2278.28   557.2 2313.14
   581.3 2324.43     617  2339.2   677.8 2370.71   794.4 2441.99   828.2 2464.94
#Mann= 4, -1 ,  0
       0     0.1       0     300    0.06       0  393.28   0.045       0
  424.71     0.1       0
#XS Ineff= 2 , 0
                          434.75         2285.89
Permanent Ineff=
       F       F
Bank Sta=393.28,424.71
XS Rating Curve= 0 ,0
Exp/Cntr=0.3,0.1

Type RM Length L Ch R = 1 ,11110   ,353.6,352.8,354.6
XS GIS Cut Line= 3
2309165.12539565667057.3631300972309253.38308774 667598.05762269
2309366.72454495667891.630577432
#Sta/Elev= 30
       0 2366.53    24.1 2352.67    32.2 2350.26    56.6 2338.12    75.7 2330.33
   101.1 2322.23   169.7 2294.65   206.5 2271.23   218.7 2266.19   234.9 2263.83
     243 2264.29   271.4 2262.86   332.2 2265.43   352.4 2265.39   357.9 2264.71
  369.62 2259.35   388.4 2258.26   398.1 2259.35   409.2 2261.33   522.6 2258.62
   538.9 2265.85   568.3 2284.22   581.2 2291.06   594.1 2296.04     637 2307.45
     697 2333.04   735.6 2350.65   790.6 2378.87   827.7 2400.79   862.5  2417.3
#Mann= 6, -1 ,  0
       0     0.1       0     290    0.06       0  369.62   0.045       0
   398.1     0.1       0     490    0.06       0  587.85     0.1       0
#XS Ineff= 2 , 0
                          409.42         2266.69
Permanent Ineff=
       F       F
Bank Sta=369.62,398.1
XS Rating Curve= 0 ,0
Exp/Cntr(USF)=0,0
Exp/Cntr=0.3,0.1

Type RM Length L Ch R = 1 ,10757   ,190.8,192.9,195.6
XS GIS Cut Line= 3
2308901.68578689667129.8874574542308969.25062224667658.368557655
2309064.92980596667989.301643017
#Sta/Elev= 30
       0  2384.8    11.4 2377.36    55.7 2353.64   152.5 2305.06   229.1 2259.02
   245.3 2258.26   265.4 2259.48   297.7    2256   366.2 2254.91   406.6 2254.93
   434.8 2257.75   441.4 2256.73   450.9 2252.03   467.1 2253.65   484.3 2251.77
   503.4 2250.35   511.9 2251.74   515.5 2254.93   523.5 2265.72   527.6 2269.68
   535.7 2275.35     544 2283.27   552.4 2288.12     569 2291.28   640.8 2310.91
   702.3 2330.48   740.9 2346.32   805.5  2377.2     823 2383.79   877.3 2407.82
#Mann= 5, -1 ,  0
       0     0.1       0     210    0.06       0     310     0.1       0
   484.3   0.045       0   511.9     0.1       0
#XS Ineff= 2 , 0
          435.81 2263.36
Permanent Ineff=
       F       F
Bank Sta=484.3,511.9
XS Rating Curve= 0 ,0
Exp/Cntr=0.3,0.1

Type RM Length L Ch R = 1 ,10564   ,46.9,47.4,49.1
XS GIS Cut Line= 6
2308714.80298688667154.2573980962308770.91893257667485.845879776
 2308775.0822413667555.2343584752308770.22504779  667639.1944177
2308723.04088227667678.051965771 2308804.7200404667980.562765315
#Sta/Elev= 30
       0    2400    51.5 2368.68    59.6  2365.2   104.2 2339.39   164.9  2308.6
   192.9 2292.28   249.9 2253.65   287.4  2253.9   330.7 2251.01   404.1 2249.55
   432.1 2251.45   436.1 2250.97  443.012246.824   462.9 2245.23  471.272246.822
   480.3 2249.41   520.1 2250.55   543.9 2254.66   552.8 2256.91   557.1 2261.99
   562.8 2265.55   622.3 2287.17   638.9 2296.12   651.3 2298.03   684.5 2299.68
     701 2307.58   721.8 2314.65   788.1 2340.63   816.7 2356.57   866.1 2380.51
#Mann= 7, -1 ,  0
       0     0.1       0   283.8    0.06       0  386.99     0.1       0
  443.01   0.045       0  471.27     0.1       0  483.49    0.06       0
  712.79     0.1       0
#XS Ineff= 2 , 0
          431.97 2258.97
Permanent Ineff=
       F       F
Bank Sta=443.01,471.27
XS Rating Curve= 0 ,0
Exp/Cntr=0.3,0.1

Type RM Length L Ch R = 1 ,10517   ,269.1,269.4,267.3
XS GIS Cut Line= 6
2308667.96576376667143.0164645472308724.08170945667474.604946227
2308728.24501817667543.9934249262308723.38782467667627.953484151
2308676.20365915667666.8110322222308757.88281727667969.321831766
#Sta/Elev= 30
       0 2408.16    89.6  2354.7   111.5 2342.51   168.2 2313.46   192.5 2298.28
     237 2265.95   261.3 2253.25   301.8 2251.07   423.4 2249.56   453.72246.098
   459.3 2245.13   479.6 2244.87  483.952246.099   490.5 2248.18   502.1 2248.15
   536.2 2251.73   552.8  2254.1   567.5 2258.23   584.1 2259.86   592.5 2266.76
   596.7 2268.88     634 2281.18   655.8 2290.99     663 2292.74   687.8  2293.7
     692 2295.24   704.4  2302.8     779  2328.4   828.7 2349.75   866.1 2369.72
#Mann= 9, -1 ,  0
       0     0.1       0   303.8    0.06       0  396.99     0.1       0
   453.7   0.045       0  483.95     0.1       0  500.52    0.06       0
  514.81     0.1       0  622.79    0.06       0  722.79     0.1       0
Bank Sta=453.7,483.95
XS Rating Curve= 0 ,0
Exp/Cntr=0.3,0.1

Type RM Length L Ch R = 1 ,10248   ,478.9,501.2,509
XS GIS Cut Line= 4
2308487.67524027667212.7703356452308461.43887413667556.498063768
2308450.48127251667708.6684362632308438.95253242 667852.46412932
#Sta/Elev= 30
       0 2343.95    20.5 2331.99    76.6 2303.47    96.7 2287.55   104.7 2280.01
   116.7 2272.33   126.9 2262.47   136.8  2254.6   144.8 2249.59   152.9 2246.24
   160.9 2245.06   204.9 2246.03   269.2 2244.63   297.3 2246.84   329.4 2244.83
   361.5 2246.79   369.5 2245.26  376.98 2240.15   385.5  2238.9   400.3 2240.12
   409.6 2243.19   473.7 2245.91   485.8 2244.74   493.8 2245.81   509.8 2252.11
   537.9 2268.11   551.9 2273.37   602.1 2284.72   626.2 2288.22   641.5 2288.31
#Mann= 5, -1 ,  0
       0     0.1       0     130    0.06       0  376.98   0.045       0
   400.3    0.06       0  424.73     0.1       0
Bank Sta=376.98,400.3
XS Rating Curve= 0 ,0
Exp/Cntr=0.3,0.1

Type RM Length L Ch R = 1 ,9746    ,225.9,212.9,206.5
XS GIS Cut Line= 5
2308289.26000888 667128.471559892308207.05136833 667286.44110448
2308044.24602135667502.4402776942307965.26124906667554.022169805
2307878.21680612667739.394594579
#Sta/Elev= 30
       0 2338.38    19.1 2327.44   108.1 2282.72   127.1  2271.3   163.1 2246.86
   181.5 2239.11   231.6 2240.92   266.7 2240.32   276.7 2239.61   289.2 2235.81
   299.4  2234.7   382.2 2233.97     447 2234.98     463 2233.93  480.242230.513
   496.4 2229.29  513.182230.514   520.3 2234.39   542.9 2233.61   549.1 2234.84
   555.1 2238.32   573.7 2253.21   585.2 2259.57   590.6 2261.83   603.8 2264.35
   630.3 2272.13   639.2  2273.2   661.3 2279.76   674.5 2285.44   747.7 2321.65
#Mann= 5, -1 ,  0
       0     0.1       0     130    0.06       0  248.08     0.1       0
  480.24   0.045       0  513.18     0.1       0
Bank Sta=480.24,513.18
XS Rating Curve= 0 ,0
Exp/Cntr(USF)=0,0
Exp/Cntr=0.3,0.1

Type RM Length L Ch R = 1 ,9533    ,38.9,36.1,36.9
XS GIS Cut Line= 4
2308082.16027118667000.5891321392307949.79400066667165.225303028
2307813.76983651667480.7030564282307727.09059292667685.444238998
#Sta/Elev= 30
       0 2334.19      11 2328.52    52.1 2311.44    92.9 2291.72   118.1 2277.98
     165  2244.1   175.5 2237.65   185.5 2232.99   255.1 2233.03   282.4 2228.46
     294 2227.64   398.1 2229.06  417.652225.672     429 2224.66  451.552225.672
   524.8 2228.33   546.6 2229.52     551  2230.5   559.4 2238.55   568.3 2245.09
   580.8 2252.71   602.2 2262.83   614.4 2264.69   641.8 2278.68   655.2 2283.53
   663.9 2288.82   681.5 2296.39   742.1 2317.17   755.1 2319.82   777.1 2327.81
#Mann= 5, -1 ,  0
       0     0.1       0     180    0.06       0  291.25     0.1       0
  417.65   0.045       0  451.55     0.1       0
#XS Ineff= 2 , 0
          388.08 2238.03
Permanent Ineff=
       F       F
Bank Sta=417.65,451.55
XS Rating Curve= 0 ,0
Exp/Cntr=0.3,0.1

Type RM Length L Ch R = 1 ,9497    ,461.1,466.5,471.2
XS GIS Cut Line= 4
2308049.97734264 666985.484386262307917.61107212667150.120557149
2307781.58690797667465.5983105492307694.90766438667670.339493119
#Sta/Elev= 30
       0 2328.45    41.2 2309.51    81.7 2287.89   130.6  2265.7   143.3 2258.25
   168.9 2240.24   181.6 2233.46   211.2 2231.41     239 2231.52   248.1 2232.73
   253.8 2232.59   288.6 2226.33   403.4 2228.73   423.7 2227.84  434.062224.376
   436.7  2223.4   447.2  2223.2   458.5 2223.42  462.522224.378   467.4 2226.51
   487.6 2226.45     519    2228     563 2234.95   567.4 2236.97   595.2 2256.25
   606.5 2260.27   615.2 2266.84   654.3 2286.15   693.3 2301.32   777.1 2329.19
#Mann= 5, -1 ,  0
       0     0.1       0     200    0.06       0  311.25     0.1       0
  434.06   0.045       0  462.52     0.1       0
#XS Ineff= 2 , 0
          400.38  2236.3
Permanent Ineff=
       F       F
Bank Sta=434.06,462.52
XS Rating Curve= 0 ,0
Exp/Cntr=0.3,0.1

Type RM Length L Ch R = 1 ,9031    ,500.4,490.9,485.4
XS GIS Cut Line= 4
     2307794.062      666768.0862307618.92292492666924.475455646
2307445.09250031667103.0489995932307209.34264322667425.667674143
#Sta/Elev= 30
       0 2321.57    30.4 2305.52    55.9 2294.24   160.8 2257.28   175.8 2249.54
   193.8 2237.22   217.8 2222.92   263.7 2221.93     308 2217.52   380.9  2216.5
     420 2217.46  430.672212.525   449.4 2211.41   460.82212.522   475.8 2224.65
   479.6 2226.18   531.2  2234.1     552 2241.16   574.9 2243.74   600.8 2253.02
   621.2 2254.82   652.2 2264.88   682.2 2272.28   699.7 2281.39   729.6  2302.6
   735.2 2304.73   754.2 2307.06   801.1 2329.31   817.8 2331.34   883.6 2363.68
#Mann= 5, -1 ,  0
       0     0.1       0     120    0.06       0   264.8     0.1       0
  430.67   0.045       0   460.8     0.1       0
Bank Sta=430.67,460.8
XS Rating Curve= 0 ,0
Exp/Cntr=0.3,0.1

Type RM Length L Ch R = 1 ,8540    ,484.7,488.8,491.3
XS GIS Cut Line= 4
2307321.45784483666373.1798943122307111.32506215666604.551981167
2307031.60193413666889.5402214692306921.17731572667227.574946484
#Sta/Elev= 30
       0 2287.18   176.5 2236.62   204.2 2224.88   226.9 2210.32   230.3 2209.47
   275.6 2207.84   302.6 2208.64   329.8 2206.73   346.4 2207.66   392.1 2204.91
   487.6 2207.16   537.5 2205.14  546.482202.995     559 2201.68  577.082202.994
   583.2 2204.45     604 2204.51   608.1 2207.81   616.5    2219   629.1 2231.04
   664.8 2256.85   679.6  2264.8   693.4 2267.43   763.8 2292.66   818.5 2307.57
   836.1 2314.28     848 2321.08   860.6 2322.04   912.2 2350.15   964.1 2373.12
#Mann= 6, -1 ,  0
       0     0.1       0     240    0.06       0     280     0.1       0
  462.55    0.06       0  546.48   0.045       0  577.08     0.1       0
#XS Ineff= 2 , 0
           471.9 2223.94
Permanent Ineff=
       F       F
Bank Sta=546.48,577.08
XS Rating Curve= 0 ,0
Exp/Cntr=0.3,0.1

Type RM Length L Ch R = 1 ,8051    ,438.1,444.8,451.3
XS GIS Cut Line= 4
2306809.84868338 666159.746366772306637.57121718666581.640449382
2306568.45672371666710.1828715982306470.79163323667019.680701597
#Sta/Elev= 30
       0 2258.09    36.1 2246.53   109.6 2216.51   143.5 2205.83   170.1 2199.66
   221.9 2197.06   239.2 2197.84   256.5  2196.3   321.3 2197.86   355.8 2194.49
   433.6 2194.65   450.9 2196.46   468.8 2195.23   482.4 2191.88   509.3 2194.55
  518.062192.299     546 2192.29   555.1 2191.63   564.2 2193.73   580.5 2194.04
   586.9 2195.41   598.2 2203.23     609 2212.23   617.4 2217.34   663.5 2255.26
   684.5 2268.29   692.9 2270.33     718 2283.49   839.7 2341.79   926.2 2387.41
#Mann= 5, -1 ,  0
       0     0.1       0     210    0.06       0     320     0.1       0
  518.06   0.045       0     546     0.1       0
#XS Ineff= 2 , 0
          450.94 2211.17
Permanent Ineff=
       F       F
Bank Sta=518.06,546
XS Rating Curve= 0 ,0
Exp/Cntr=0.3,0.1

Type RM Length L Ch R = 1 ,7606    ,589.8,581,569.7
XS GIS Cut Line= 4
2306513.78784566665953.1844618162306387.55667828666280.389312221
2306260.77851221666370.3994533092306179.81697577 666780.69278083
#Sta/Elev= 30
       0 2267.54    42.9  2256.2   132.9 2229.87   152.8 2220.44   184.3 2199.57
   210.1 2188.83   251.8 2191.08   326.1 2189.63   347.3 2188.82     359 2186.97
   379.7  2187.7   386.6 2186.63  392.74 2182.55   403.9 2181.19412.30772182.561
   428.3 2184.75   454.1 2183.92   476.4 2184.92   492.2 2183.58     509 2185.88
   684.3 2185.33   688.4 2186.42   692.5 2189.12   704.7 2200.24   737.3 2222.61
   786.3 2253.02     827 2269.45   843.3 2274.75   866.6 2279.37   924.4 2288.17
#Mann= 4, -1 ,  0
       0     0.1       0     220    0.06       0  392.74   0.045       0
412.3077     0.1       0
#XS Ineff= 2 , 0
                          510.37         2188.59
Permanent Ineff=
       F       F
Bank Sta=392.74,412.3077
XS Rating Curve= 0 ,0
Exp/Cntr=0.3,0.1

Type RM Length L Ch R = 1 ,7025    ,602,609.9,613.2
XS GIS Cut Line= 4
2305862.72740163665726.9658090362305775.03769686665959.139434675
2305805.41621067666459.8919184542305762.63742983666716.876904518
#Sta/Elev= 30
       0 2239.86    53.7 2226.32   160.6 2196.25   216.2 2187.73   270.1 2175.04
   302.3 2170.42   330.4    2173   466.5 2176.35   477.9 2175.93   490.7 2172.86
   538.8 2172.78   549.7 2171.68   573.4 2171.68   590.8 2173.43   630.9 2172.05
     667 2172.84     695 2175.33     699 2175.23   707.1 2171.77   711.1 2171.31
   735.1 2174.38   743.1 2178.56     759 2191.64   779.5 2206.35   803.4 2219.55
   840.4 2237.07   852.9 2239.96     891 2255.25   970.1 2291.85  1010.4  2312.1
#Mann= 5, -1 ,  0
       0     0.1       0  348.18    0.06       0  448.18     0.1       0
   549.7   0.045       0   573.4     0.1       0
#XS Ineff= 2 , 0
          467.01  2192.2  692.88         2190.24
Permanent Ineff=
       F       F
Bank Sta=549.7,573.4
XS Rating Curve= 0 ,0
Exp/Cntr=0.3,0.1

Type RM Length L Ch R = 1 ,6415    ,235.3,249.5,265.6
XS GIS Cut Line= 4
2305438.23170187665665.4439136842305324.71579744666059.920660454
2305230.10243832666289.2226534982305110.41849184666615.724494295
#Sta/Elev= 30
       0 2222.17    53.8 2210.49    78.8 2202.36    91.3 2195.57   101.8 2194.29
   117.8 2188.59   178.7  2178.5     212 2175.35   237.4  2165.4   245.3 2163.57
   278.6 2164.29   455.1 2161.86   476.2 2160.19   537.3 2159.53   543.1 2156.92
   554.6 2155.55   565.72156.924   584.9 2160.31     614 2160.27   632.5 2162.56
   649.8 2177.59   679.8  2197.5   688.3 2200.56   692.6 2203.81   701.1 2206.09
   718.1 2214.96   803.2 2250.77   909.8 2301.46   931.2  2309.8  1006.3 2344.33
#Mann= 5, -1 ,  0
       0     0.1       0     410    0.06       0  520.48     0.1       0
   543.1   0.045       0   565.7     0.1       0
#XS Ineff= 2 , 0
          487.14  2166.3
Permanent Ineff=
       F       F
Bank Sta=543.1,565.7
XS Rating Curve= 0 ,0
Exp/Cntr=0.3,0.1

Type RM Length L Ch R = 1 ,6166    ,81.1,72.9,73.3
XS GIS Cut Line= 6
2305327.48981728665695.5278955032305286.63425227666112.640726772
2305140.90268561666119.4819322752304967.39887628666187.770603586
2304904.67446708666187.7706035862304831.82767738666549.677038944
#Sta/Elev= 30
       0 2216.91    41.9 2206.85    49.9 2203.55      65 2201.25    98.1 2190.88
   118.2 2182.69   146.3 2177.75   178.5 2174.98     212 2162.55   226.7  2160.1
   258.9 2161.76   307.1 2161.08   355.3 2162.52     595 2156.86   653.5 2157.31
  668.972152.742   703.3 2151.94  714.79 2152.74   729.9 2156.72   761.4 2157.09
   789.7 2161.11   816.8 2160.47   879.3 2196.05   903.4 2207.48     915 2214.57
   928.4 2217.39  1067.2 2286.34  1091.6 2297.56  1103.9 2301.27    1186  2334.3
#Mann= 6, -1 ,  0
       0     0.1       0     370    0.06       0  668.97   0.045       0
  714.79     0.1       0  751.87    0.06       0  886.82     0.1       0
Bank Sta=668.97,714.79
XS Rating Curve= 0 ,0
Exp/Cntr(USF)=0,0
Exp/Cntr=0.3,0.1

Type RM Length L Ch R = 1 ,6093    ,224.5,217.6,201.7
XS GIS Cut Line= 6
 2305291.0236668665660.2909411062305250.16810179666077.403772375
2305104.43653513666084.244977878 2304930.9327258 666152.53364919
 2304868.2083166 666152.53364919 2304795.3615269666514.440084548
#Sta/Elev= 30
       0 2225.64    37.1 2218.77    81.3 2207.53    89.3 2204.14   101.4 2203.92
   141.6 2190.73   149.6 2184.12   153.6  2182.5   185.8 2175.78     230 2171.61
   266.2 2159.73   318.6 2161.43   517.5 2159.43   565.9 2155.15   602.8 2156.41
   690.7  2155.6   720.12151.264   743.4 2149.98  752.812151.264   772.4 2155.38
   837.8 2156.17   862.4 2168.12   904.4 2191.32   935.8 2205.77   952.1 2211.48
   964.4 2219.26   976.6  2221.7   984.8 2227.61  1115.3    2294    1186 2323.71
#Mann= 9, -1 ,  0
       0     0.1       0     300    0.06       0   717.4     0.1       0
   720.1   0.045       0  752.81     0.1       0  773.56    0.06       0
  809.71     0.1       0  826.82    0.06       0  926.82     0.1       0
Bank Sta=720.1,752.81
XS Rating Curve= 0 ,0
Exp/Cntr(USF)=0,0
Exp/Cntr=0.3,0.1

Type RM Length L Ch R = 1 ,5875    ,293.2,295.8,299.9
XS GIS Cut Line= 4
2304876.83806018 665616.091030092304813.23227328665897.233096063
2304714.41811412 666156.480682572304671.28029358666493.765634861
#Sta/Elev= 30
       0 2222.05    50.3 2209.12    66.7 2208.49   214.4 2187.47   247.2 2177.65
   288.2 2160.14   309.6 2149.55   335.3 2148.04   347.9 2149.99   416.6 2149.61
   455.1 2150.28   459.5 2150.09  467.55 2147.78   476.5 2146.08  492.742147.781
   509.1 2150.89   536.5  2152.3   553.6 2151.95   570.4 2161.55   618.8 2180.64
     643  2191.8   663.2 2199.19   687.4 2209.64   699.5 2213.02   715.6 2219.41
   723.7 2223.47   731.7 2224.56   785.9 2253.65   860.8 2298.82   905.7 2322.89
#Mann= 7, -1 ,  0
       0     0.1       0      30    0.06       0      50     0.1       0
  467.55   0.045       0  492.74     0.1       0  565.69    0.06       0
  665.69     0.1       0
#XS Ineff= 2 , 0
          346.91    2161
Permanent Ineff=
       F       F
Bank Sta=467.55,492.74
XS Rating Curve= 0 ,0
Exp/Cntr=0.3,0.1

Type RM Length L Ch R = 1 ,5579    ,549.6,532.3,523.6
XS GIS Cut Line= 4
2304644.13466071665542.5926724672304577.76575395665812.156329465
 2304455.0755108665972.6101154052304448.66654035666445.460863846
#Sta/Elev= 30
       0 2233.29    35.6 2226.43    80.9 2212.54   130.4 2201.71   146.8 2200.47
   183.9 2189.73   216.9 2177.54   262.2 2168.71   277.6 2162.39     289 2151.79
   293.7 2148.61   304.1 2145.45   359.4 2142.63   385.6 2141.66  393.162142.592
   399.7 2145.22   427.9 2144.44   496.2 2146.38   524.2 2144.76   574.6 2145.09
   612.2 2146.09   640.2 2149.71   664.2    2149   676.2  2153.5   688.2  2160.4
   727.7 2179.05   765.2  2193.7   856.2 2235.06   889.6 2251.42   952.5 2285.25
#Mann= 6, -1 ,  0
       0     0.1       0   359.4   0.045       0  393.16     0.1       0
  447.61    0.05       0   569.6    0.07       0   669.6     0.1       0
#XS Ineff= 2 , 0
                          478.87         2159.33
Permanent Ineff=
       F       F
Bank Sta=359.4,393.16
XS Rating Curve= 0 ,0
Exp/Cntr=0.3,0.1

Type RM Length L Ch R = 1 ,5047    ,135,136.5,138.8
XS GIS Cut Line= 4
2304052.23421218665470.5664219442304020.38139992665771.409601505
2304065.94064273666016.5298076592304152.14273719 666396.35094877
#Sta/Elev= 30
       0  2242.7    26.8 2232.39    54.9 2218.54      75 2210.75   131.3 2200.99
   183.6 2189.82   235.2 2169.67   276.1 2158.13   288.2 2151.37   304.3  2138.5
   308.4  2137.1     345 2136.62  365.242132.751     385 2131.66   392.1 2132.75
   397.9 2136.63     402 2137.72   430.4 2135.34   485.7 2136.08     520 2138.97
   564.8 2144.98   622.2 2149.52   655.1 2149.75   684.6 2157.13   741.2 2161.51
   757.6 2169.69   810.9 2190.89     856 2203.92   888.8 2215.39   941.3 2231.51
#Mann= 9, -1 ,  0
       0     0.1       0  365.24   0.045       0   392.1     0.1       0
  392.52    0.06       0  492.52    0.05       0  601.84    0.06       0
  641.84    0.07       0  701.84    0.05       0  801.84     0.1       0
#XS Ineff= 2 , 0
          336.78 2147.81
Permanent Ineff=
       F       F
Bank Sta=365.24,392.1
XS Rating Curve= 0 ,0
Exp/Cntr=0.3,0.1

Type RM Length L Ch R = 1 ,4911    ,37.4,34.5,34.8
XS GIS Cut Line= 6
2303892.67137432665457.264434617 2303781.3933923665732.886265186
2303838.84272464665758.9995980682303889.76372376665806.003597254
2303900.20905691665849.0905965082303905.43172349666389.636587152
#Sta/Elev= 30
       0 2227.75    47.4 2213.95    81.9  2198.4   103.4 2190.84     125 2187.32
   150.9 2180.94   215.6 2153.88   225.7  2147.7   245.8 2144.61     263 2136.74
   280.3 2132.33   335.4 2131.31     470 2133.67  486.612130.524   502.1 2128.92
  514.932130.527   522.1 2134.28   590.1 2134.16   642.1 2132.03   710.1 2132.36
   726.1 2135.43   738.1 2134.53   766.1 2135.62   786.1 2139.31     810 2150.36
     822    2154   834.1  2162.9   878.1 2189.46   926.1 2215.75  1014.6 2256.28
#Mann= 4, -1 ,  0
       0     0.1       0  486.61   0.045       0  514.93    0.06       0
  682.39     0.1       0
#XS Ineff= 2 , 0
          432.79 2181.56
Permanent Ineff=
       F       F
Bank Sta=486.61,514.93
XS Rating Curve= 0 ,0
Exp/Cntr(USF)=0,0
Exp/Cntr=0.3,0.1

Type RM Length L Ch R = 1 ,4876    ,296.7,305,307.9
XS GIS Cut Line= 6
2303859.48308006665476.5218399272303748.20509804665752.143670496
2303805.65443038665778.257003378 2303856.5754295665825.261002564
2303867.02076265665868.3480018182303872.24342923666408.893992462
#Sta/Elev= 30
       0 2214.94    13.6 2211.97    78.4 2189.26   112.9 2182.11   169.1 2159.82
   181.3 2152.48   201.2 2150.01   246.6 2132.88   358.7 2130.87   450.1 2133.85
  461.122130.159   466.6  2128.6  491.112130.157   494.8 2132.66   498.8 2133.46
   526.9 2132.16   554.9  2133.9   594.9 2131.63   672.7 2131.03   718.9 2133.79
   726.9 2132.95   738.9 2135.37   770.9 2147.43   786.9 2155.01   798.9 2162.48
   806.9 2163.46   829.9 2178.01   866.9 2198.78   926.9 2227.45  1014.6 2266.66
#Mann= 7, -1 ,  0
       0     0.1       0  327.24    0.06       0  347.24     0.1       0
  461.12   0.045       0  491.11    0.06       0  572.39    0.05       0
  662.39     0.1       0
#XS Ineff= 2 , 0
          432.11 2210.05
Permanent Ineff=
       F       F
Bank Sta=461.12,491.11
XS Rating Curve= 0 ,0
Exp/Cntr(USF)=0,0
Exp/Cntr=0.3,0.1

Type RM Length L Ch R = 1 ,4571    ,547.3,549.5,545
XS GIS Cut Line= 4
2303693.86631505665396.9086842812303598.32799885665729.782335051
2303510.00747474666062.5412316822303457.24031908666303.021159876
#Sta/Elev= 30
       0  2229.6   129.3 2176.24   141.8 2168.44   158.4 2167.98   166.7 2163.38
   187.5 2156.36   233.3  2146.3   279.1 2133.38   295.7 2130.06   341.1  2129.3
     354 2126.67   386.8 2127.31   411.9 2125.35   422.8 2126.45   458.8 2125.16
  486.072125.156   494.8 2128.03   643.7 2124.64   664.4 2122.76   668.5 2123.83
   689.2 2137.79   723.1 2168.55   734.6 2177.46   742.4 2180.47   762.9 2183.96
   818.6 2200.85   869.4 2225.17   902.1  2244.8   918.5 2251.83   936.8 2257.14
#Mann= 5, -1 ,  0
       0     0.1       0   458.8   0.045       0  486.07     0.1       0
  486.31    0.06       0  686.31     0.1       0
#XS Ineff= 2 , 0
          420.06 2136.86
Permanent Ineff=
       F       F
Bank Sta=458.8,486.07
XS Rating Curve= 0 ,0
Exp/Cntr=0.3,0.1

Type RM Length L Ch R = 1 ,4022    ,454.9,455.4,455.4
XS GIS Cut Line= 4
2303336.23958108665257.5923170632303099.26606587665584.931185687
2303047.37397747665921.0806073782303017.39606587666235.903281105
#Sta/Elev= 30
       0 2209.26    28.4 2200.95   127.9 2178.65     202 2167.88   260.4 2151.17
   320.5 2138.26   412.5 2123.75  428.43 2114.53   432.7  2113.2   444.8 2112.91
  454.27 2114.52     461 2116.28   473.2 2115.33   505.5 2116.63   522.7 2114.15
   537.9 2113.71   550.1 2116.14   687.7 2117.34     716 2116.21   736.2 2118.35
   748.4  2126.2   769.3 2145.73   808.6 2175.18   816.7 2178.29   832.7 2179.84
     885 2199.93  1025.6 2263.05  1041.7 2265.07  1049.7    2270  1060.5 2273.76
#Mann= 6, -1 ,  0
       0     0.1       0  428.43   0.045       0  454.27     0.1       0
  484.11    0.05       0  584.11    0.06       0  684.11     0.1       0
#XS Ineff= 2 , 0
                          687.14         2131.51
Permanent Ineff=
       F       F
Bank Sta=428.43,454.27
XS Rating Curve= 0 ,0
Exp/Cntr=0.3,0.1

Type RM Length L Ch R = 1 ,3566    ,567.1,582.4,579.1
XS GIS Cut Line= 4
2302764.54787632665155.3600645622302664.65484268665482.469662929
2302620.83797483665872.0540133062302624.59273598 666166.41511791
#Sta/Elev= 30
       0 2225.08      37 2214.35   110.8  2189.7     211 2164.57   219.4  2160.1
   231.9 2157.25   286.9 2134.62   315.7 2125.07   340.7 2119.28   344.6 2117.62
   358.2 2106.64   364.9 2105.12  373.352106.617     381 2108.17   401.1 2107.12
   457.5 2108.39   517.8 2106.86   598.5 2106.94   630.5 2108.81   715.1    2107
   735.2 2108.85   746.4 2114.02   780.4 2135.35   815.2 2150.98   827.2 2157.88
   839.2 2160.27   847.2 2166.68   922.3 2205.51   971.2 2233.41  1028.4  2269.4
#Mann= 6, -1 ,  0
       0     0.1       0   358.2   0.045       0  373.35     0.1       0
  432.02    0.05       0  632.02    0.06       0  824.06     0.1       0
#XS Ineff= 2 , 0
                          631.74         2119.14
Permanent Ineff=
       F       F
Bank Sta=358.2,373.35
XS Rating Curve= 0 ,0
Exp/Cntr=0.3,0.1

Type RM Length L Ch R = 1 ,2984    ,377.4,382.7,386.3
XS GIS Cut Line= 4
2302345.14407945 665165.944251732302227.06212039665497.781298022
2302167.42645063665804.3837910552302189.85991649666120.779358556
#Sta/Elev= 30
       0 2206.46    50.1 2191.74   125.4 2165.41   181.7 2151.58   262.4 2136.12
   334.6 2111.26     368 2102.32   408.7 2099.13   547.2 2097.91   571.7 2099.05
   583.9 2097.82  593.972093.711   612.4 2092.23  622.482093.713   627.1 2095.71
   636.9 2103.46   640.9 2105.31   661.3 2106.17   673.4  2117.2     681 2122.13
   737.2 2145.78   813.7 2181.91   821.8 2187.19   825.8 2188.87   833.8 2189.61
   837.8 2191.77     842 2195.68   958.1 2253.25   973.1 2261.32   981.8  2267.4
#Mann= 6, -1 ,  0
       0     0.1       0     220    0.05       0  522.22     0.1       0
  593.97   0.045       0  622.48    0.06       0  724.57     0.1       0
Bank Sta=593.97,622.48
XS Rating Curve= 0 ,0
Exp/Cntr(USF)=0,0
Exp/Cntr=0.3,0.1
